--- UPTROUTRN.prj (project) ---

Proj Title=UPTROUTRN
Current Plan=p01
Default Exp/Contr=0,0
English Units
Geom File=g01
Flow File=f01
Plan File=p01
BEGIN DESCRIPTION:
----------MODEL BY WOOD PLC 2022----------
AFH study
Randolph County, WV
HEC-RAS Version: RAS 6.2
Vertical Datum: NAVD88
Projection: NAD 1983 StatePlane West Virginia S FIPS 4702 (US Feet)
Terrain: 1-meter LIDAR (FEMA Region III 3DEP collected 2016-2018)
Land Use: 2019 NLCD
Hydrologic Method:
WV SIR2010-5033 regression equations
Additional Model Notes:
None
END DESCRIPTION:
DSS Export Rating Curves= 0
DSS Export Rating Curve Sorted= 0
DSS Export Volume Flow Curves= 0
DXF OffsetX= 0
DXF OffsetY= 0
DXF ScaleX= 0
DXF ScaleY= 0

--- UPTROUTRN.p01 (plan) ---

Plan Title=Floodplain
Program Version=6.20
Short Identifier=Floodplain
Geom File=g01
Flow File=f01
Subcritical Flow
K Sum by GR= 0
Std Step Tol= 0.01
Critical Tol= 0.01
Num of Std Step Trials= 20
Max Error Tol= 0.3
Flow Tol Ratio= 0.001
Split Flow NTrial= 30
Split Flow Tol= 0.02
Split Flow Ratio= 0.02
Log Output Level= 0
Friction Slope Method= 1
Unsteady Friction Slope Method= 2
Unsteady Bridges Friction Slope Method= 1
Parabolic Critical Depth
Global Vel Dist= 0 , 0 , 0
Global Log Level= 0
CheckData=True
Encroach Param=-1 ,0,0, 0
Mapping Interval=1HOUR
Computation Time Step Use Courant=        0
Computation Time Step Use Time Series=    0
Computation Time Step Count To Double=0
Computation Time Step Max Doubling=0
Computation Time Step Max Halving=0
Computation Time Step Residence Courant=0
Run HTab= 0
Run UNet= 0
Run Sediment= 0
Run PostProcess= 0
Run WQNet= 0
Run RASMapper=-1
UNET Theta= 0
UNET Theta Warmup= 0
UNET ZTol= 0
UNET ZSATol= 0
UNET MxIter= 0
UNET Max Iter WO Improvement= 0
UNET MaxInSteps= 0
UNET DtIC= 0
UNET DtMin= 0
UNET MaxCRTS= 0
UNET WFStab= 0
UNET SFStab= 0
UNET WFX= 1
UNET SFX= 1
UNET Gravity=32.174
UNET 1D Methodology=Finite Difference
UNET DSS MLevel= 1
UNET Pardiso=0
UNET DZMax Abort= 0
UNET Use Existing IB Tables= 0
UNET Froude Reduction=False
UNET Froude Limit= 0
UNET Froude Power= 0
UNET D1 Cores= 0
UNET WindReference=Eulerian
UNET WindDragFormulation=Hsu (1988)
UNET D2 Coriolis=0
UNET D2 Cores= 0
UNET D2 Theta= 1
UNET D2 Theta Warmup= 1
UNET D2 Z Tol= 0.01
UNET D2 Volume Tol= 0.01
UNET D2 Max Iterations= 20
UNET D2 Equation= 0
UNET D2 RampUpFraction=0.1
UNET D2 TimeSlices= 1
UNET D2 Turbulence Formulation=Non-Conservative (original)
UNET D2 Eddy Viscosity=0.3
UNET D2 Transverse Eddy Viscosity=0.1
UNET D2 Smagorinsky Mixing=0
UNET D2 BCVolumeCheck=0
UNET D2 Cores=0
UNET D2 SolverType=PARDISO (Direct)
UNET D2 Minimum Iterations= 2147483647
UNET D2 Maximum Iterations= 2147483647
UNET D2 Restart Number= 10
UNET D2 Relaxation Coeff=1.3
UNET D2 SOR Precondition Iterations= 10
UNET D2 ILUT Maximum Fill= 8
UNET D2 ILUT Tolerance=1E-08
UNET D1D2 MaxIter= 0
UNET D1D2 ZTol=0.01
UNET D1D2 QTol=0.1
UNET D1D2 MinQTol=1
Write IC File= 0
Write IC File at Fixed DateTime=0
Write IC File at Sim End=0
Echo Input=False
Echo Parameters=False
Echo Output=False
Write Detailed= 0
HDF Write Warmup=0
HDF Write Time Slices=0
HDF Flush=0
HDF Compression= 1
HDF Chunk Size= 1
HDF Spatial Parts= 1
HDF Use Max Rows=0
HDF Fixed Rows= 1
Calibration Method= 0
Calibration Iterations= 20
Calibration Max Change=0.05
Calibration Tolerance=0.2
Calibration Maximum=1.5
Calibration Minimum=0.5
Calibration Optimization Method= 1
WQ AD Non Conservative
WQ ULTIMATE=-1
WQ Max Comp Step=1HOUR
WQ Output Interval=15MIN
WQ Output Selected Increments= 0
WQ Output face flow=0
WQ Output face velocity=0
WQ Output face area=0
WQ Output face dispersion=0
WQ Output cell volume=0
WQ Output cell surface area=0
WQ Output cell continuity=0
WQ Output cumulative cell continuity=0
WQ Output face conc=0
WQ Output face dconc_dx=0
WQ Output face courant=0
WQ Output face peclet=0
WQ Output face adv mass=0
WQ Output face disp mass=0
WQ Output cell mass=0
WQ Output cell source sink temp=0
WQ Output nsm pathways=0
WQ Output nsm derived pathways=0
WQ Create Restart=0
WQ Fixed Restart=0
WQ System Summary=0
WQ Write To DSS=0
Sorting and Armoring Iterations= 10
XS Update Threshold= 0.02
Bed Roughness Predictor= 0
Hydraulics Update Threshold= 0.02
Energy Slope Method= 1
Volume Change Method= 1
Sediment Retention Method= 0
Sediment TS Multiplier= 1
Warm Up Method= 0
XS Weighting Method= 0
Number of US Weighted Cross Sections= 1
Number of DS Weighted Cross Sections= 1
Upstream XS Weight=0
Main XS Weight=1
Downstream XS Weight=0
Number of DS XS's Weighted with US Boundary= 1
Upstream Boundary Weight= 1
Weight of XSs Associated with US Boundary= 0
Number of US XS's Weighted with DS Boundary= 1
Downstream Boundary Weight= 0.5
Weight of XSs Associated with DS Boundary= 0.5
Percentile Method= 0
Sediment Output Level= 3
Mass or Volume Output= 0
Output Increment Type= 1
Profile and TS Output Increment= 1
Transport Output Increment 1
XS Output Flag= 0
XS Output Increment= 10
Read HDF5 Sediment Hotstart= 0
Sediment Hotstart Type= 0
Write Gradation File= 0
Read Gradation Hotstart= 0
Write HDF5 File= 1
Write Binary Output= 1
Write DSS Sediment File= 0
DSS Sediment Output Type= 1
SV Curve= 0
Specific Gage Flag= 0
Subcell Erosion Methods= 0
Subcell Deposition Methods= 0
Advection Scheme= 1
Matrix Solver= 0
Implicit Weighting Factor= 1
Maximum Outer Loop Convergence Iterations= 5
Convergence Maximum Absolute= 0.001
Convergence RMSE= 0.0001
Grain Fractions Max Abs Error= 0.001
Max Subgrid Regions= 1
Max Subgrid Length Scale= 3.402823E+38
Initial Layer Thickness= 3.402823E+38
Min Layer Thickness= 3.402823E+38
Max Layer Thickness= 3.402823E+38
Number of Layers= 5

--- UPTROUTRN.f01 (steady flow) ---

Flow Title=Flow
Program Version=6.20
Number of Profiles= 1
Profile Names=P100yr
River Rch & RM=UPTROUTRN,Main            ,9360
     484
River Rch & RM=UPTROUTRN,Main            ,3947
     655
River Rch & RM=UPTROUTRN,Main            ,2291
     730
Boundary for River Rch & Prof#=UPTROUTRN,Main            , 1
Up Type= 0
Dn Type= 3
Dn Slope=0.03137
DSS Import GetInterval= 0
DSS Import GetPeak= 0
DSS Import FillOption= 0

--- UPTROUTRN.g01 (geometry) ---

Geom Title=Geometry
Program Version=6.20

River Reach=UPTROUTRN       ,Main
Reach XY= 30
     2193591.218      615029.245     2193763.006      615155.634
     2193705.367      615405.982     2193822.728      615518.829
     2193752.242      615698.343     2193791.305      615913.187
     2193593.344      616533.247     2193626.331      616743.317
     2193572.641      617575.739      2193771.86      617667.405
     2193880.193      617918.447     2194015.892      618014.367
     2194032.559      618210.895      2194268.67      618418.881
      2194356.17      618691.103      2194649.92      619076.867
     2194663.462      619260.548     2194748.184      619390.409
     2195101.597      619647.941     2195012.204      620041.432
     2195072.068      620157.476     2195008.393      620468.117
      2194703.81      621184.626        2194914.      621347.735
     2195187.168      621401.836     2195343.271      621531.139
2195723.92121674621600.894963877     2196048.514      621937.572
     2196135.849      622108.478     2196391.699       622150.34

Type RM Length L Ch R = 1 ,9360    ,347.8,360.2,372.2
XS GIS Cut Line= 4
  2193461.802606615183.7675660552193565.23987493615114.372351735
 2193693.9731407 614837.228094072193657.54147621614681.079945392
#Sta/Elev= 30
       0 2552.81    26.6 2542.02    41.1 2538.56    55.8 2533.21   113.6 2518.09
   131.5 2515.68   172.8 2514.51   187.6 2510.86   199.9 2512.12  206.172510.548
     212 2509.42   216.32510.548     227 2514.46   231.7 2515.15   258.2 2513.03
   284.3  2513.4   302.4  2516.7   328.8 2518.41   337.6 2517.09   350.8 2517.13
   356.5 2518.56   387.9 2520.96   410.8 2523.92   430.2 2524.43   463.1  2536.1
   491.8  2550.3   504.1 2553.99   516.4 2560.77     537  2569.4   590.5  2595.4
#Mann= 7 ,-1,0
       0      .1       0     110     .06       0  206.17    .045       0
   216.3     .06       0  284.56      .1       0  334.56     .12       0
  394.56      .1       0
Bank Sta=206.17,216.3
XS Rating Curve= 0 ,0
Exp/Cntr=0.3,0.1

Type RM Length L Ch R = 1 ,9000    ,335.9,335.9,333.6
XS GIS Cut Line= 5
2193524.88315596615323.9037552712193679.88230864615265.372606708
 2193757.5943551615315.5785220522193857.36376401615317.922110339
2193974.79560745615275.584607253
#Sta/Elev= 30
       0 2552.48    24.9 2541.49    59.1 2528.55    72.9 2525.22    84.8 2523.85
   106.1 2518.29   123.2 2514.65   144.6 2512.02   161.7 2509.09   180.2 2507.33
   189.8 2507.37   197.6 2506.15   206.3 2502.75   218.4 2495.45   221.92494.056
   231.7 2493.02   238.72494.067   252.5 2496.31   260.8 2496.07   284.8 2497.89
   300.8 2496.75   316.8 2496.76   320.8 2496.04   328.7 2497.65   363.9 2500.37
   370.2  2502.5     378 2507.08   390.8 2509.81   437.5  2515.7   482.8 2520.18
#Mann= 5 ,-1,0
       0      .1       0   221.9    .045       0   238.7      .1       0
  255.68     .06       0     458      .1       0
#XS Ineff= 2 , 0
                         256.067            2500
Permanent Ineff=
       F       F
Bank Sta=221.9,238.7
XS Rating Curve= 0 ,0
Exp/Cntr(USF)=0,0
Exp/Cntr=0.3,0.1

Type RM Length L Ch R = 1 ,8664    ,266.4,262.2,255
XS GIS Cut Line= 4
2193565.80662949615524.4537615952193764.43468761615535.381285382
2193958.44721939 615644.74116221 2194082.7614997615644.630149159
#Sta/Elev= 30
       0 2547.32    26.4 2535.51    54.5 2524.43    98.5 2511.01   110.5 2509.01
   138.6 2499.97   158.6 2498.59   178.6 2495.22   186.7 2492.77   198.9 2485.07
   207.8 2484.29   218.9 2486.32  242.03 2482.74     250 2481.88  257.592482.739
   262.9 2486.83   267.5 2487.91   290.5 2488.18   322.6 2485.85     341 2485.81
   350.2 2487.16   382.1 2486.74   414.4  2488.9   435.4 2498.08   451.8 2508.11
   467.4 2513.89   479.4 2516.91   511.9 2529.47   527.4 2533.76     546 2541.71
#Mann= 5 ,-1,0
       0      .1       0  242.03    .045       0  257.59      .1       0
  258.93     .06       0  408.93      .1       0
Bank Sta=242.03,257.59
XS Rating Curve= 0 ,0
Exp/Cntr=0.3,0.1

Type RM Length L Ch R = 1 ,8401    ,356.9,356.5,359.1
XS GIS Cut Line= 5
2193559.19172658615716.5699281772193638.86650592615760.968025268
2193763.87734918615807.053494448 2193864.1470356615786.733392984
 2194015.6668667615860.477879039
#Sta/Elev= 30
       0  2527.1    33.5 2509.54    51.2 2502.79      79 2484.24    89.4 2479.01
    92.6  2478.4     108 2479.64     131 2478.54   143.8 2479.46   160.9 2478.48
   176.5 2476.11   194.9 2478.17   207.5 2476.25   224.7  2477.7     2462474.159
   253.3 2473.16   261.92474.181   273.7 2477.32     290 2483.25   294.1 2483.87
   314.5 2483.91   326.8 2487.25   343.6 2486.03   350.6 2486.69   387.2  2500.2
   430.3 2508.67   451.3 2516.19   469.1 2521.46   486.9 2529.09   495.3 2531.86
#Mann= 5 ,-1,0
       0      .1       0     246    .045       0   261.9      .1       0
  314.45     .06       0  426.75      .1       0
#XS Ineff= 2 , 0
          221.88 2490.68
Permanent Ineff=
       F       F
Bank Sta=246,261.9
XS Rating Curve= 0 ,0
Exp/Cntr=0.3,0.1

Type RM Length L Ch R = 1 ,8045    ,235.5,244.4,248.1
XS GIS Cut Line= 3
2193452.58012156616061.9135895442193637.53240223616137.609003518
 2193926.5047886616132.686046381
#Sta/Elev= 30
       0 2507.04    12.5 2503.85    21.2 2502.74    68.7 2490.91    81.7 2488.67
   124.9 2483.25   164.7 2479.81   185.4 2479.19   214.7 2475.87   222.5 2474.06
   234.3  2469.8   246.5 2466.77  253.342463.954   261.9  2463.3   271.3 2463.99
   282.5 2464.95   306.5 2463.34   314.5 2463.61   318.5 2465.28   326.5 2470.11
   334.5 2473.65   350.5  2484.7   354.5 2485.63   366.5 2486.42   378.5 2486.19
   402.5 2499.74   418.5 2504.45   446.5 2511.54   474.3 2520.55   488.9  2526.3
#Mann= 5 ,-1,0
       0      .1       0  253.34    .045       0   271.3      .1       0
  319.84     .06       0  419.84      .1       0
Bank Sta=253.34,271.3
XS Rating Curve= 0 ,0
Exp/Cntr=0.3,0.1

Type RM Length L Ch R = 1 ,7800    ,216.7,211.5,205.8
XS GIS Cut Line= 4
2193415.40822994616286.4159760882193601.84077722 616323.26892148
2193716.73525403616407.8139138492193867.39876607616413.233464642
#Sta/Elev= 30
       0 2507.88      13 2503.42    33.4 2497.95    90.5 2484.52   115.4 2480.13
   127.2 2477.28   135.3 2474.63   143.5 2474.02   151.6 2472.51     163 2471.45
     172 2469.96   180.2 2466.85   188.3 2462.18   192.9 2460.09   195.9 2459.45
   212.8  2458.2   257.5 2458.28   262.5 2458.04  268.552456.406   277.4  2455.7
  288.372456.407   296.1 2459.97   298.9 2460.61   307.2 2461.11   322.1 2460.69
   340.1 2466.37   404.2 2484.52   456.2 2497.47     476 2503.32483.4496 2504.85
#Mann= 5 ,-1,0
       0      .1       0  268.55    .045       0  288.37      .1       0
  372.69     .06       0  472.69      .1       0
Bank Sta=268.55,288.37
XS Rating Curve= 0 ,0
Exp/Cntr(USF)=0,0
Exp/Cntr=0.3,0.1

Type RM Length L Ch R = 1 ,7589    ,330.8,330.8,329.8
XS GIS Cut Line= 3
2193411.37343806616505.682710505 2193520.2418162616559.457866699
2193843.96615971616583.352311792
#Sta/Elev= 30
       0 2497.21    14.3 2492.08    32.1 2487.97    74.9 2474.51   112.4 2464.74
   129.4 2462.27   137.4 2462.89   157.5 2461.61   165.5 2461.96   177.5 2459.89
   181.5 2456.96   185.5 2453.15  189.95  2450.2   193.6 2449.48   201.6  2449.4
  210.182450.201   231.3 2452.85   249.7 2450.56   276.1  2453.1   293.8 2452.74
   301.8 2456.87   307.8 2458.29   309.9 2458.65   317.9 2457.06   321.9 2457.64
   329.9 2460.92   337.9 2465.68     374 2479.37   418.2 2491.26     446 2499.77
#Mann= 5 ,-1,0
       0      .1       0  189.95    .045       0  210.18      .1       0
  261.43     .06       0  351.43      .1       0
Bank Sta=189.95,210.18
XS Rating Curve= 0 ,0
Exp/Cntr=0.3,0.1

Type RM Length L Ch R = 1 ,7258    ,259.2,260.1,259.4
XS GIS Cut Line= 3
2193373.13573376616837.0423366452193465.26809724616878.230922671
2193808.86761751616890.153934416
#Sta/Elev= 30
       0 2485.96    14.5 2481.24    26.6 2476.42    55.9 2466.17      69 2460.82
    78.1 2457.82   100.8 2444.55   107.8 2441.75   111.8 2441.23   119.8  2441.1
   135.8 2441.29   147.9 2442.47   171.9 2441.78   191.9  2442.4   195.9 2442.16
  203.63 2438.94     211 2438.55   223.9 2438.92   239.9 2439.33   243.9 2440.51
   247.9 2440.87   259.9 2439.42   271.9  2439.5   287.9  2447.6     312 2453.51
     384 2473.47   400.6  2479.1     416  2485.6     428  2488.5444.7264 2493.66
#Mann= 5 ,-1,0
       0      .1       0  190.92     .06       0  203.63    .045       0
   223.9     .06       0  290.92      .1       0
Bank Sta=203.63,223.9
XS Rating Curve= 0 ,0
Exp/Cntr(USF)=0,0
Exp/Cntr=0.3,0.1

Type RM Length L Ch R = 1 ,6998    ,234.9,236.3,235.7
XS GIS Cut Line= 3
2193282.08728044617099.3485950212193375.30355408617125.362438827
2193766.59512132617150.292372474
#Sta/Elev= 30
       0 2479.01    39.5 2467.89    97.7 2454.73   129.7 2448.14   162.1 2442.45
   173.8 2438.71   177.8 2437.06   185.8 2432.27   189.8  2430.7   193.8  2429.8
   222.1 2431.03   241.9 2430.94     294 2432.71   302.1 2431.85  309.152429.049
   318.1 2428.14   322.1 2428.16   325.62429.049   330.1 2430.73   342.1 2431.28
   346.2 2432.09   350.2 2435.72   354.2 2440.04     359 2442.32   374.2 2446.95
   394.3 2450.04   418.3 2455.68   450.4 2465.27   481.8 2476.24 488.863 2479.14
#Mann= 5 ,-1,0
       0      .1       0  309.15    .045       0   325.6      .1       0
  376.78     .06       0  476.78      .1       0
#XS Ineff= 2 , 0
        297.1779    2435
Permanent Ineff=
       F       F
Bank Sta=309.15,325.6
XS Rating Curve= 0 ,0
Exp/Cntr(USF)=0,0
Exp/Cntr=0.3,0.1

Type RM Length L Ch R = 1 ,6762    ,84,78.3,70.1
BEGIN DESCRIPTION:
Structure XS 4
END DESCRIPTION:
XS GIS Cut Line= 4
2193243.17258656617382.8649816862193473.72259647617366.424058095
2193666.40912713  617374.46447172193780.35019747617346.351586557
#Sta/Elev= 30
       0 2485.47    33.1 2473.28    69.9 2460.82    97.2 2452.95   111.5 2449.52
   121.3 2448.25   145.4 2441.95   153.4 2441.59   182.2 2436.72   209.5 2434.52
   221.6 2432.92   229.6 2431.21   241.6 2426.46   245.6 2425.46   269.6 2424.03
   281.6 2420.84     313 2420.58   317.7 2420.28   320.7 2420.58   339.9 2422.24
   369.7 2422.27   381.7 2424.65   421.8 2427.34   429.4 2430.58     443 2439.15
   450.5 2442.99   495.8 2454.49     529 2467.66     537  2471.5   541.3 2472.86
#Mann= 5 ,-1,0
       0      .1       0  311.14     .06       0     313    .045       0
   320.7     .06       0  411.14      .1       0
#XS Ineff= 2 , 0
                          339.64         2424.87
Permanent Ineff=
       F       F
Bank Sta=313,320.7
XS Rating Curve= 0 ,0
Exp/Cntr=0.5,0.3

Type RM Length L Ch R = 1 ,6684    ,41.4,42.9,45.2
BEGIN DESCRIPTION:
Structure XS 3
END DESCRIPTION:
XS GIS Cut Line= 6
 2193283.3345256617684.691474033 2193535.6700522617570.905343845
2193529.56099497617480.0929250382193561.58736262617432.771726106
2193575.13008705617396.3659520952193783.23880095 617349.66042114
#Sta/Elev= 30
       0 2502.03     8.5 2498.02    18.5 2496.51    62.4 2477.89    75.9 2473.93
   106.1 2461.94     115 2457.45   124.3 2456.59   163.3 2441.56   181.7 2435.82
   220.3 2417.54   224.7 2416.36   281.3 2415.94   323.1 2417.19   358.9 2416.26
   389.9 2417.78  401.58 2414.62   409.5 2413.71  417.03 2414.62   427.3 2418.19
     438 2419.85   463.6 2420.82   469.6 2421.94   494.2 2421.64   506.5 2423.68
   555.7 2427.43   563.9 2430.97   584.4 2442.96   629.5 2454.24   677.7 2473.21
#Mann= 4 ,-1,0
       0      .1       0  401.58    .045       0  417.03     .06       0
  544.43      .1       0
#XS Ineff= 2 , 0
          389.68 2424.32
Permanent Ineff=
       F       F
Bank Sta=401.58,417.03
XS Rating Curve= 0 ,0
Exp/Cntr(USF)=0,0
Exp/Cntr=0.5,0.3

Type RM Length L Ch R = 1 ,6641    ,118.3,115.8,115.7
BEGIN DESCRIPTION:
Structure XS 2
END DESCRIPTION:
XS GIS Cut Line= 6
  2193296.949182617712.6648991582193564.31920379617592.657598545
2193558.21014656617501.8451797382193590.23651421617454.523980806
2193603.77923864617418.1182067952193790.11385605617373.486399315
#Sta/Elev= 30
       0 2502.97     7.9 2501.27    26.3  2492.5    38.4 2488.88    82.5 2470.41
     117 2457.97   125.7 2453.38   135.2 2452.49   152.6 2445.02   187.7  2432.9
   218.4 2416.53   235.9 2415.13   268.4 2415.03   277.4 2413.02   293.1 2412.07
   390.1 2414.57  398.94 2413.28   406.9 2413.27   428.7 2420.08   456.1 2426.32
   468.9 2426.71   478.6 2425.39   485.2  2426.6   501.7  2425.1   518.1 2425.91
   530.5 2427.83   563.4  2439.3   607.9 2449.67   625.1 2454.79   672.3 2473.26
#Mann= 5 ,-1,0
       0      .1       0     290     .06       0  398.94    .045       0
   406.9     .06       0  530.69      .1       0
#XS Ineff= 2 , 0
          389.68 2418.64
Permanent Ineff=
       F       F
Bank Sta=398.94,406.9
XS Rating Curve= 0 ,0
Exp/Cntr(USF)=0,0
Exp/Cntr=0.5,0.3

Type RM Length L Ch R = 1 ,6525    ,237.2,245.2,246.6
BEGIN DESCRIPTION:
Structure XS 1
END DESCRIPTION:
XS GIS Cut Line= 4
2193313.73745707617736.1458131852193509.81680476617666.883954052
2193702.96959501617492.2660275062193804.42358586617435.685917228
#Sta/Elev= 30
       0 2500.67    32.3 2486.75      45 2482.31    76.3 2469.46    87.4 2465.27
   100.2 2461.38   123.4 2452.58   134.1 2447.68   154.7 2443.45   167.2 2437.45
   189.1 2430.44   210.8 2420.01     225 2414.74   228.4 2414.01   265.1 2414.16
   275.8 2411.56     293 2411.04  301.142409.384   305.9 2408.24  314.922409.385
   335.4 2412.67   378.3  2414.1   395.4 2415.56   423.2 2423.94   448.4 2429.35
   468.3 2435.26   478.9  2437.3   515.5 2446.27   571.5 2463.09584.5005 2468.32
#Mann= 5 ,-1,0
       0      .1       0  267.95     .06       0  301.14    .045       0
  314.92     .06       0  417.95      .1       0
Bank Sta=301.14,314.92
XS Rating Curve= 0 ,0
Exp/Cntr(USF)=0,0
Exp/Cntr=0.3,0.1

Type RM Length L Ch R = 1 ,6280    ,236.8,242.3,242.7
XS GIS Cut Line= 3
2193406.86699902617907.9189003862193681.93336299617790.458128743
2193913.88121586617595.681406146
#Sta/Elev= 30
       0 2491.95    14.5 2485.95    27.5 2482.13    84.1 2461.75   140.2 2440.04
   188.4 2425.44   284.1 2405.77   292.8 2405.07     302 2402.49   327.1 2401.65
   338.6 2396.61   350.8 2393.75   378.3 2398.46   395.3 2400.36   416.9 2398.84
   423.7 2397.14   432.6 2396.41   454.4 2397.12   463.9 2399.93   475.2 2398.63
   495.3 2399.96     511 2403.69   520.2 2409.78   531.6 2415.13   547.5 2426.94
     558 2433.08   568.5 2442.07   574.8 2446.43   594.5 2457.35601.9786 2459.99
#Mann= 5 ,-1,0
       0      .1       0   389.1     .06       0   423.7    .045       0
   454.4     .06       0   519.1      .1       0
#XS Ineff= 2 , 0
        399.9375    2405
Permanent Ineff=
       F       F
Bank Sta=423.7,454.4
XS Rating Curve= 0 ,0
Exp/Cntr(USF)=0,0
Exp/Cntr=0.3,0.1

Type RM Length L Ch R = 1 ,6037    ,385.1,386.2,385
XS GIS Cut Line= 2
2193603.37134175618136.1320812212194042.95079847617789.465646725
#Sta/Elev= 30
       0 2460.19    17.7 2451.87    39.7 2446.47    97.8    2427   123.3 2420.19
   140.4 2413.73   162.2 2407.38   179.3 2404.28   196.3 2404.02   245.5 2397.66
   261.9 2393.98   296.5 2392.68   306.7  2390.6   327.1 2390.52   338.8  2389.1
  345.622386.671   352.5 2385.75  360.322386.671     390 2389.64   398.4 2389.15
     410 2386.88   418.5 2387.55   439.1 2396.08   455.5 2408.35   469.8 2414.03
   482.8 2423.62   492.5 2429.53     521 2442.94   530.8 2448.41   559.8 2461.28
#Mann= 5 ,-1,0
       0      .1       0     320     .06       0  345.62    .045       0
  360.32     .06       0     440      .1       0
Bank Sta=345.62,360.32
XS Rating Curve= 0 ,0
Exp/Cntr=0.3,0.1

Type RM Length L Ch R = 1 ,5651    ,271.9,271.5,269
XS GIS Cut Line= 2
2193812.94664375 618380.791817792194250.93094739618071.533677639
#Sta/Elev= 30
       0 2448.29    10.6 2443.79    23.5 2440.16    52.9  2429.7    76.7 2419.36
    96.8 2412.31   116.6 2403.78     146 2395.11   165.6 2383.95   180.2 2378.69
   188.6 2378.06   234.1  2380.2   243.9 2378.89   262.9 2378.66  269.692374.754
   276.7  2373.7  287.382374.754   297.5 2376.63   309.1 2377.36   339.1 2376.47
   355.1 2376.91   373.8 2382.57   390.8 2385.42   395.7 2387.25   420.2  2401.6
   444.6 2419.78   458.4  2426.9   493.6 2447.26   512.9 2455.29   536.2 2463.22
#Mann= 4 ,-1,0
       0      .1       0  269.69    .045       0  287.38     .06       0
     290      .1       0
#XS Ineff= 2 , 0
                           307.1         2392.61
Permanent Ineff=
       F       F
Bank Sta=269.69,287.38
XS Rating Curve= 0 ,0
Exp/Cntr=0.3,0.1

Type RM Length L Ch R = 1 ,5380    ,210.6,220.4,232.4
XS GIS Cut Line= 3
2193968.08547963618599.0537008172194273.04578184618368.118606518
2194376.22635626618280.595388997
#Sta/Elev= 30
       0 2436.75     9.7 2433.83    21.4  2428.5    35.7 2424.06    80.4 2404.13
    95.9 2396.37   115.7  2382.5   120.5 2379.71   142.2 2370.19   156.1 2369.27
   221.8 2369.05   268.1 2371.92   295.5 2369.73   315.5 2370.54   329.8  2369.9
   335.5 2369.23   341.6 2367.16   346.9 2366.78   351.3 2367.34   356.4  2369.4
   371.4 2381.39   381.2 2387.35   391.9 2395.87   395.4 2397.71   444.3 2416.58
   474.8  2430.5   487.9 2435.66   504.6 2443.89   511.7 2445.27   517.8 2447.71
#Mann= 4 ,-1,0
       0      .1       0     220     .06       0   341.6    .045       0
   351.3      .1       0
#XS Ineff= 2 , 0
          317.98 2371.24
Permanent Ineff=
       F       F
Bank Sta=341.6,351.3
XS Rating Curve= 0 ,0
Exp/Cntr=0.3,0.1

Type RM Length L Ch R = 1 ,5159    ,41.9,42.7,41
XS GIS Cut Line= 4
 2194035.0296992618696.1586846082194277.12945462 618521.09319754
2194402.56652739618672.1615995382194605.24526207 618535.62013617
#Sta/Elev= 30
       0 2436.72      31  2424.1    63.1 2414.46    90.3 2404.88   100.7 2399.76
   124.8 2385.39   146.2 2375.43   160.5 2371.24   169.2    2370     192 2369.15
   203.8 2367.36   228.5 2368.27   257.9 2368.04     285 2365.33   306.7 2365.67
   347.4 2364.54   376.9 2362.06   384.9 2360.59  396.88 2362.02   411.8 2364.09
   460.1 2360.59   495.1 2359.09   501.3 2360.24   518.6 2360.34     526  2361.9
   550.1 2375.16   645.4 2413.71   697.3 2432.02   714.1 2436.72   739.5 2445.62
#Mann= 5 ,-1,0
       0      .1       0     260     .06       0   376.9    .045       0
  396.88     .06       0  545.12      .1       0
#XS Ineff= 2 , 0
                          409.53         2373.55
Permanent Ineff=
       F       F
Bank Sta=376.9,396.88
XS Rating Curve= 0 ,0
Exp/Cntr(USF)=0,0
Exp/Cntr=0.3,0.1

Type RM Length L Ch R = 1 ,5116    ,130.8,120.2,109.1
XS GIS Cut Line= 4
2194048.94932154618708.8903837382194269.74583532618548.311100986
2194395.18290809618699.3795029842194613.19997676618550.908224297
#Sta/Elev= 30
       0 2435.06     7.8 2433.26    28.7 2424.28    58.4 2414.81    90.9 2400.46
   142.4 2375.69   149.1 2373.06   162.3 2369.59   173.9  2368.2   191.1 2367.94
   199.7 2366.44   241.4 2367.49   264.7 2365.42   276.8 2365.84   289.7 2364.65
   346.9 2363.99   357.7  2362.9   369.82359.945   388.72359.976     402 2362.44
   445.7 2359.63   487.5 2357.98     519 2360.81   544.3 2375.04     577 2389.59
   586.7 2392.48   595.5 2394.15     698 2433.76   727.1 2444.42   733.1 2445.74
#Mann= 7 ,-1,0
       0      .1       0     120     .05       0     160      .1       0
     240     .06       0   369.8    .045       0   388.7     .06       0
  529.37      .1       0
#XS Ineff= 2 , 0
                          403.56        2368.727
Permanent Ineff=
       F       F
Bank Sta=369.8,388.7
XS Rating Curve= 0 ,0
Exp/Cntr(USF)=0,0
Exp/Cntr=0.3,0.1

Type RM Length L Ch R = 1 ,4996    ,427.6,427.3,427
XS GIS Cut Line= 2
2194193.84720582618886.4864080782194627.86298668618552.343739876
#Sta/Elev= 30
       0 2422.46       8 2420.13    19.7 2413.51    41.5 2403.93    74.3 2391.59
   124.1 2379.15   150.9 2368.36   172.6 2363.19   185.1 2357.98   192.3 2357.17
   199.4 2358.76   231.6 2359.66  241.992357.014   250.3 2356.02  255.922357.014
   262.1 2359.03   290.7 2357.13   310.6 2359.81     321 2360.25   330.6 2364.03
   353.4 2376.82   370.5 2383.32   376.5 2384.66   395.6 2392.37   452.2 2417.85
   467.4 2421.76   500.5  2435.2   512.8  2438.1   527.9 2444.06   547.7 2449.94
#Mann= 6 ,-1,0
       0     .05       0      70      .1       0     190     .06       0
  241.99    .045       0  255.92     .06       0     310      .1       0
#XS Ineff= 2 , 0
        232.2967    2361
Permanent Ineff=
       F       F
Bank Sta=241.99,255.92
XS Rating Curve= 0 ,0
Exp/Cntr=0.3,0.1

Type RM Length L Ch R = 1 ,4569    ,346.4,346.6,343.1
XS GIS Cut Line= 2
2194456.57971775619237.1585187222194866.94899589618872.881442108
#Sta/Elev= 30
       0 2400.48    42.1 2383.37    63.6 2377.45      79 2369.87    90.4 2368.34
     113 2358.81   138.5 2351.13   156.6 2347.61   186.7 2344.72     235 2345.78
   243.4 2344.52     249    2344  255.05 2344.51   265.1 2346.37   285.9 2346.09
   289.2 2347.67   295.2 2354.41     300 2357.53     315 2358.62   319.9 2362.71
   325.5 2369.73   331.2 2372.38   427.8 2401.34   448.7  2411.1   475.5 2420.91
   486.2 2426.42   498.4  2429.2     521 2439.23   532.4 2441.14548.7264 2446.86
#Mann= 5 ,-1,0
       0      .1       0     240     .06       0   243.4    .045       0
  255.05     .06       0     380      .1       0
#XS Ineff= 2 , 0
                           276.5         2360.58
Permanent Ineff=
       F       F
Bank Sta=243.4,255.05
XS Rating Curve= 0 ,0
Exp/Cntr(USF)=0,0
Exp/Cntr=0.3,0.1

Type RM Length L Ch R = 1 ,4222    ,278.4,275.2,271.4
XS GIS Cut Line= 3
2194657.89613562      619466.7562195017.12036217 619143.48727045
2195053.31534636619052.771619157
#Sta/Elev= 30
       0  2388.7    46.1 2374.31    56.9 2368.95    67.6 2364.71    94.5 2350.74
      99 2347.01  109.782334.702   110.7 2334.05     116 2333.94  128.562334.706
   211.6 2337.75   226.5 2337.43   247.5 2340.44   259.5 2343.03   297.3 2346.78
   317.1 2346.48   336.9 2353.57   348.3 2356.61   382.3 2368.89   401.3 2377.97
     412 2379.29   420.9  2384.5   447.4 2395.19   475.7 2403.47   496.6 2408.43
   507.3    2410   511.6 2411.56   541.7  2424.8   573.6 2440.88   580.9 2445.22
#Mann= 5 ,-1,0
       0      .1       0  109.78    .045       0  128.56      .1       0
     250     .06       0     370      .1       0
#XS Ineff= 2 , 0
                          172.68         2356.57
Permanent Ineff=
       F       F
Bank Sta=109.78,128.56
XS Rating Curve= 0 ,0
Exp/Cntr=0.3,0.1

Type RM Length L Ch R = 1 ,3947    ,143.5,147.2,149.9
XS GIS Cut Line= 4
2194753.47989811619667.1300370172194926.90552349619621.364941433
2195052.15736403619361.2265033752195101.53549348619105.905443799
#Sta/Elev= 30
       0 2401.38    19.3 2393.32    79.1 2373.05   143.4 2345.04   155.9 2341.17
   172.4 2332.41   179.4 2330.11   219.5 2329.62   237.3  2328.1   259.5 2329.26
  266.15 2327.83   274.5 2326.56  282.96 2327.83   302.2 2328.69     335 2332.99
   370.5 2334.13   383.8 2333.64   420.2 2341.49   441.2 2342.84   450.4 2345.29
   468.1 2346.03   478.2 2350.43   488.5 2351.16     492 2352.29     517 2364.21
     533 2370.55   602.6 2393.62   684.1 2410.09   700.4 2415.34728.1358 2426.87
#Mann= 5 ,-1,0
       0      .1       0  266.15    .045       0  282.96      .1       0
  319.36     .06       0  528.08      .1       0
#XS Ineff= 2 , 0
          212.56 2334.56
Permanent Ineff=
       F       F
Bank Sta=266.15,282.96
XS Rating Curve= 0 ,0
Exp/Cntr(USF)=0,0
Exp/Cntr=0.3,0.1

Type RM Length L Ch R = 1 ,3800    ,21.2,21.2,21.1
XS GIS Cut Line= 6
2194759.28762178619707.5034134872194934.11430566 619649.23067598
2195068.49657621619635.2579846432195125.60496653619567.559547246
2195172.13722964619474.4950210312195368.74127683619544.604868399
#Sta/Elev= 30
       0 2403.67      22 2395.32    51.5 2386.17    81.6 2374.78   106.3 2364.46
   144.3 2346.62   169.6    2339   194.3 2329.09   286.5 2325.22   325.4 2326.58
   330.5 2325.97  333.84 2323.92   336.9 2322.49   340.7 2322.27   345.8 2323.94
   350.9    2327   389.1 2331.09   454.8 2331.78   523.2 2334.74   532.5 2334.11
   544.4  2331.3   554.4 2333.69   563.8 2334.52     570 2337.12   578.4 2343.83
   582.7 2344.55     606 2355.02   625.1 2355.73   629.5 2356.84   723.4 2390.56
#Mann= 9 ,-1,0
       0      .1       0  279.56     .06       0  333.84    .045       0
   345.8     .06       0  373.27     .07       0  420.25     .06       0
   494.4      .1       0  574.68     .06       0  684.68      .1       0
Bank Sta=333.84,345.8
XS Rating Curve= 0 ,0
Exp/Cntr=0.3,0.1

Type RM Length L Ch R = 1 ,3779    ,162.6,167.8,172.9
XS GIS Cut Line= 6
 2194772.4087719619724.0699823132194947.23545578619665.797244806
2195081.61772633619651.8245534692195138.72611665619584.126116071
2195185.25837976619491.0615898562195362.74181319619554.127000577
#Sta/Elev= 30
       0 2399.42    52.7 2383.99    67.2 2376.84    96.7  2364.9   130.5  2348.7
   176.8 2334.68   193.2 2328.25   257.2  2325.7   329.1 2326.25   334.52323.372
   338.6 2321.91  345.81 2323.38   356.1 2325.34   380.1 2324.64   389.8 2329.98
   393.2 2330.27   413.1  2330.3   436.9 2327.37   488.6 2330.07   514.7 2333.34
     522 2330.63   526.3 2330.61   534.3 2333.26   543.7 2333.68   549.9 2336.54
   560.2 2346.56   571.9 2349.41   585.7 2355.12   606.9  2355.9     703 2390.27
#Mann= 7 ,-1,0
       0      .1       0  269.56     .06       0   334.5    .045       0
  345.81     .06       0   504.4      .1       0  544.68     .06       0
  664.68      .1       0
#XS Ineff= 2 , 0
          287.07 2335.83  377.41         2334.14
Permanent Ineff=
       F       F
Bank Sta=334.5,345.81
XS Rating Curve= 0 ,0
Exp/Cntr=0.3,0.1

Type RM Length L Ch R = 1 ,3611    ,234.2,235.3,236
XS GIS Cut Line= 4
 2194764.3189997619820.081803839 2194963.0358621619781.542775978
2195205.10913085619824.8991823212195405.03033788619812.855736115
#Sta/Elev= 30
       0 2406.76    40.6 2391.24    63.8 2383.95    93.6 2372.85   126.2 2358.11
   138.4 2354.28   175.1 2338.73   207.6 2322.75   215.8 2321.59   244.2 2321.85
   268.6 2320.47   309.2 2320.74  317.742319.123   325.5    2318  336.032319.124
   341.7 2321.79   344.4 2321.94   410.8 2321.64     419 2322.94   435.2 2329.66
   463.4 2331.95   483.5 2331.42   515.5 2346.35   535.6 2353.04   551.6 2359.98
   607.7 2375.57   619.7 2380.39   627.7 2380.99   639.5 2386.04648.6284 2387.96
#Mann= 8 ,-1,0
       0      .1       0     170     .06       0  272.42      .1       0
  317.74    .045       0  336.03      .1       0  372.42     .06       0
  478.34      .1       0  568.34     .12       0
#XS Ineff= 2 , 0
          244.62 2329.65  369.76          2334.2
Permanent Ineff=
       F       F
Bank Sta=317.74,336.03
XS Rating Curve= 0 ,0
Exp/Cntr(USF)=0,0
Exp/Cntr=0.3,0.1

Type RM Length L Ch R = 1 ,3376    ,341.9,344.5,341.2
XS GIS Cut Line= 2
2194762.79082833619956.7122674562195381.07869799620130.844917601
#Sta/Elev= 30
       0 2396.58    30.5 2383.21    59.9 2372.24   101.2 2355.36   117.8 2347.47
   130.3 2343.39   146.9 2336.15   163.6 2325.25   184.3 2313.43   192.6 2312.32
   209.2 2314.81   221.7 2314.11   234.2 2315.37   247.9 2314.72   254.4 2312.89
   259.1 2312.24   270.6 2312.89   279.9 2314.74     309 2313.64   321.4 2315.46
   446.1 2315.34   462.7 2317.84   491.8 2319.35     496 2322.13   504.1 2330.92
   520.9 2351.31     525 2354.93   533.5 2360.04   587.4  2384.7   642.3 2403.13
#Mann= 7 ,-1,0
       0      .1       0   254.4    .045       0   270.6      .1       0
     380     .06       0     490     .07       0     500     .06       0
     590      .1       0
#XS Ineff= 2 , 0
                          303.46         2328.18
Permanent Ineff=
       F       F
Bank Sta=254.4,270.6
XS Rating Curve= 0 ,0
Exp/Cntr=0.3,0.1

Type RM Length L Ch R = 1 ,3031    ,137.8,137.3,137.6
XS GIS Cut Line= 4
2194680.56741932620205.0693175522194837.51219156620299.236180894
2195138.18533416620338.8853865122195265.39320219 620395.05509447
#Sta/Elev= 30
       0 2384.62    36.9 2371.59    75.6 2352.98    88.2  2348.9   111.5 2336.79
   150.1 2320.34   189.7 2306.52   201.4 2305.24   233.5 2304.93   302.7 2307.83
   327.9  2305.7   341.9 2301.82   351.1 2300.69  371.13 2301.83   387.4 2305.17
   403.6 2305.43   411.7 2306.93   423.8  2304.5   431.8 2304.59   439.9 2307.32
     456 2309.29   484.3 2309.67   488.5 2311.84   497.2  2319.4     506 2331.75
   510.3 2336.51     526  2349.4   580.5    2375   593.4 2379.33625.3607 2392.94
#Mann= 5 ,-1,0
       0      .1       0   341.9    .045       0  371.13      .1       0
  383.03     .06       0   586.3      .1       0
Bank Sta=341.9,371.13
XS Rating Curve= 0 ,0
Exp/Cntr(USF)=0,0
Exp/Cntr=0.3,0.1

Type RM Length L Ch R = 1 ,2894    ,45.4,44.8,45.3
XS GIS Cut Line= 3
2194625.76607759620275.3900607822194780.61452917620399.456178942
2195160.62305926620494.439462576
#Sta/Elev= 30
       0  2385.6    42.8 2368.46    65.6 2357.45    92.4 2346.93   105.6 2339.66
   115.8 2334.89   126.1 2328.42   136.4 2323.61   156.6 2311.09   169.2 2304.97
   175.6 2303.02   188.4 2301.78   225.9 2303.27   247.4 2303.38   346.4 2301.51
     400 2301.48   416.5  2302.6  428.65 2298.43   441.2 2296.99     4472298.341
   449.5 2299.55   453.6 2303.14   457.7 2305.17   494.8 2306.89   498.9 2309.52
   522.7 2336.65   527.8 2340.55     569 2357.92   581.4 2361.51   590.1 2365.71
#Mann= 5 ,-1,0
       0      .1       0  428.65    .045       0     447      .1       0
  458.42     .06       0  558.42      .1       0
Bank Sta=428.65,447
XS Rating Curve= 0 ,0
Exp/Cntr(USF)=0,0
Exp/Cntr=0.3,0.1

Type RM Length L Ch R = 1 ,2849    ,171.1,173.6,175.2
XS GIS Cut Line= 3
2194609.06651782620317.1657908612194763.91496939620441.231909021
2195143.92349949620536.215192656
#Sta/Elev= 30
       0 2379.96    13.6 2375.67    55.2 2358.95    70.5 2350.32    83.2 2344.76
   118.9 2326.37   132.1 2317.41     153 2304.84   161.6 2301.62   173.1 2300.69
   201.9 2301.87   281.3 2301.99   360.2 2300.07   399.8  2300.3   421.3  2298.9
  427.23  2297.1   433.7 2295.91  446.34 2297.08   454.3 2303.64   458.4 2305.02
   474.9 2305.95   487.3 2305.55   491.4 2306.68   495.5 2310.49     512 2329.99
   516.2 2334.26   518.6 2335.68   540.9  2344.1   582.1 2362.23   590.1 2364.88
#Mann= 5 ,-1,0
       0      .1       0  388.42     .06       0  427.23    .045       0
  446.34     .06       0  478.42      .1       0
Bank Sta=427.23,446.34
XS Rating Curve= 0 ,0
Exp/Cntr(USF)=0,0
Exp/Cntr=0.3,0.1

Type RM Length L Ch R = 1 ,2675    ,384.9,384.1,383.4
XS GIS Cut Line= 3
2194553.79242411620476.8385505732194956.88449982620670.392137119
 2195112.5400669620678.685659234
#Sta/Elev= 30
       0 2357.07    33.7 2345.82    51.5 2337.63      68 2331.04    95.8  2315.9
   109.1 2309.41   126.9 2302.35   139.9 2298.89   154.9    2297   184.6 2298.31
   193.4 2296.67   205.9 2296.12   265.8 2297.62   304.8 2296.89   357.6  2297.5
   364.8 2296.55  374.042292.083   382.8 2291.06   388.7 2291.28  391.212292.083
   394.8 2293.94     402 2299.62   406.4 2301.33   428.6    2301   433.1 2303.62
   446.4 2315.44   458.5 2320.71   550.6 2345.26     586 2358.72     603  2366.3
#Mann= 5 ,-1,0
       0      .1       0  374.04    .045       0  391.21      .1       0
     420     .06       0  527.15      .1       0
Bank Sta=374.04,391.21
XS Rating Curve= 0 ,0
Exp/Cntr=0.3,0.1

Type RM Length L Ch R = 1 ,2291    ,260.7,250.9,237.5
XS GIS Cut Line= 4
2194300.35184058620990.941069113 2194513.1444307620913.025318098
2194905.06458674 621050.209816582195100.43579451620885.493272761
#Sta/Elev= 30
       0 2371.82    51.1 2360.79    97.8 2347.55   129.1  2336.3   148.9 2327.48
   166.5 2321.23   191.5 2307.15     207 2295.64   217.1 2291.99   255.2 2287.66
   318.8 2287.17   352.7 2288.96     429 2287.03     474 2284.29  485.61 2284.29
     501 2285.47   574.4 2282.99   598.5 2283.64   636.7 2280.33   640.9 2281.32
   647.6  2285.7   656.1 2287.76   724.3 2296.87   766.2 2305.56   786.7 2307.37
   809.4 2317.09   817.2 2318.05   837.8 2327.38   883.2 2341.22   897.4 2344.26
#Mann= 5 ,-1,0
       0      .1       0     474    .045       0  485.61      .1       0
  566.61     .06       0  761.84      .1       0
#XS Ineff= 2 , 0
                           584.7         2301.37
Permanent Ineff=
       F       F
Bank Sta=474,485.61
XS Rating Curve= 0 ,0
Exp/Cntr=0.3,0.1

Type RM Length L Ch R = 1 ,2040    ,250.1,246.9,239.5
XS GIS Cut Line= 3
2194571.13002983 621375.092286032194914.75647851621064.506842023
2195106.39430567 620917.47437119
#Sta/Elev= 30
       0 2345.98     8.8 2342.05    19.1 2339.06    44.6 2328.16   106.9 2310.23
   114.6 2306.35   143.7 2287.81   152.4 2283.56   163.9 2281.53   191.8 2279.65
     206 2280.85  211.16    2279   229.5 2278.51   235.5 2278.99   241.5 2279.95
   253.4  2279.3   344.8 2281.67   378.8 2280.44     395 2281.72     422 2280.77
   435.4 2281.89   459.7  2280.3   475.1 2286.36   488.4 2289.28   586.9 2304.48
   612.1 2306.92   639.5 2318.81   646.3 2319.42   666.6 2325.86704.7315 2334.74
#Mann= 5 ,-1,0
       0      .1       0  211.16    .045       0   235.5      .1       0
     360     .06       0  613.19      .1       0
#XS Ineff= 2 , 0
          205.63 2287.99428.8823            2288
Permanent Ineff=
       F       F
Bank Sta=211.16,235.5
XS Rating Curve= 0 ,0
Exp/Cntr(USF)=0,0
Exp/Cntr=0.3,0.1

Type RM Length L Ch R = 1 ,1794    ,482.9,485,486
XS GIS Cut Line= 4
2194868.10306911621556.3267722072194930.15406838621372.974636565
  2195058.032201621033.8932710582195128.56165813620996.888977331
#Sta/Elev= 30
       0 2358.05    20.2 2351.52    41.3  2342.9    96.2 2317.01   104.7 2314.95
   117.3 2309.41   162.4 2293.13   182.4 2284.23  201.832273.898   210.6 2272.59
  219.822273.896     226 2275.45   235.3 2275.79   291.7 2273.97   304.5 2275.29
   347.2 2274.03   378.1 2276.65     403 2275.43   407.1 2276.81   415.6  2282.9
   419.9 2284.51   449.5  2286.7   548.2 2301.66   557.5 2304.11   576.4 2304.96
     599 2313.33   608.1 2314.16   617.1 2317.21   630.7 2322.34   635.6 2325.27
#Mann= 5 ,-1,0
       0      .1       0  201.83    .045       0  219.82      .1       0
  303.57     .06       0  413.57      .1       0
#XS Ineff= 2 , 0
                          378.56         2286.63
Permanent Ineff=
       F       F
Bank Sta=201.83,219.82
XS Rating Curve= 0 ,0
Exp/Cntr=0.3,0.1

Type RM Length L Ch R = 1 ,1309    ,298.7,300.4,297.3
XS GIS Cut Line= 3
2195257.90988364621688.5946601162195514.89547561621288.839294835
2195576.08252132 621148.10908971
#Sta/Elev= 30
       0 2339.58     8.8 2335.06    42.1 2321.93    51.6 2319.33   115.1 2293.53
   146.7 2282.17   151.5 2279.94   166.2 2268.94  178.012262.035   184.8 2260.97
  194.732262.035   203.8    2264   275.1 2265.84   313.2 2264.06   322.5 2266.39
   346.4 2265.77   377.5  2262.5   403.5 2264.06   455.4 2264.16   470.1 2263.22
   475.2 2264.94   485.1  2272.5   492.3 2276.16     501 2283.54   514.1 2291.98
   531.6 2306.99   544.6 2314.54   570.2 2324.18     597 2336.31628.6888 2348.89
#Mann= 7 ,-1,0
       0     .06       0      30      .1       0  178.01    .045       0
  194.73      .1       0     270     .07       0     310     .06       0
     380      .1       0
#XS Ineff= 2 , 0
                          275.45         2275.38
Permanent Ineff=
       F       F
Bank Sta=178.01,194.73
XS Rating Curve= 0 ,0
Exp/Cntr(USF)=0,0
Exp/Cntr=0.3,0.1

Type RM Length L Ch R = 1 ,1008    ,77.6,78.8,82.7
XS GIS Cut Line= 3
2195451.39221957621822.950782064 2195645.2917035621600.147027246
2195781.38264563621255.704465744
#Sta/Elev= 30
       0 2345.34    50.1 2323.16      66 2305.78    69.9 2304.16    81.2 2303.52
    87.2 2304.25    92.5 2303.24   104.8 2296.42   118.1 2291.24   137.9 2284.91
   200.3 2274.22   267.5 2265.94   283.4  2260.2   298.6 2257.42  301.732256.057
   307.2 2254.57   314.1 2254.41   320.1 2254.51   326.62256.058   354.5  2256.9
   386.2 2258.97   401.8 2258.13   423.2 2259.03   429.4 2260.01   483.5 2259.66
   500.7 2260.83     505 2261.85   524.9 2269.64   605.1 2302.66665.7148 2330.45
#Mann= 7 ,-1,0
       0      .1       0      80     .06       0     210      .1       0
     260     .06       0  301.73    .045       0   326.6     .06       0
  445.36      .1       0
#XS Ineff= 2 , 0
                        385.6294            2269
Permanent Ineff=
       F       F
Bank Sta=301.73,326.6
XS Rating Curve= 0 ,0
Exp/Cntr(USF)=0,0
Exp/Cntr=0.3,0.1

Type RM Length L Ch R = 1 ,929     ,25.8,25.8,25.8
XS GIS Cut Line= 4
2195527.30239233621852.0058321532195666.52942427621673.854596436
2195768.40965224621557.5055385392195946.08809342621346.052203013
#Sta/Elev= 30
       0 2322.82    44.2 2303.82    49.3 2299.86    53.9 2294.89    59.6 2290.83
    79.7 2287.95    89.9 2288.53    99.5 2286.25   130.5 2282.17   150.8 2276.78
   228.6 2265.59   240.7 2263.15   256.1 2262.46   273.1 2259.11   296.1 2257.75
   304.3 2256.36   312.1 2253.42   321.3 2252.07  330.19 2253.39   352.5 2255.92
   402.1 2257.89   502.9 2256.23   506.6 2257.23   527.5 2271.41   543.1 2279.66
   582.4 2291.21   599.4 2297.13   610.8 2299.37   621.5 2303.56   656.9 2310.47
#Mann= 5 ,-1,0
       0     .06       0   306.1     .07       0   312.1    .045       0
  330.19     .07       0  460.75      .1       0
#XS Ineff= 2 , 0
                          358.29         2264.35
Permanent Ineff=
       F       F
Bank Sta=312.1,330.19
XS Rating Curve= 0 ,0
Exp/Cntr(USF)=0,0
Exp/Cntr=0.3,0.1

Type RM Length L Ch R = 1 ,904     ,103.1,101.7,102
XS GIS Cut Line= 4
2195547.89323154621867.6045079472195687.12026348 621689.45327223
2195789.00049145621573.1042143332195966.67893263621361.650878807
#Sta/Elev= 30
       0 2323.57    52.4 2299.92    58.9 2293.19      64 2288.77    65.4  2288.3
    79.2 2286.69     133 2275.45   170.6 2269.41   235.5 2261.95     252    2261
   270.2 2261.47   295.1 2257.24   308.52253.152   316.9 2251.92   322.2 2251.99
  326.84 2253.14   331.9 2254.66   343.4 2255.84   391.1 2256.26   406.8 2257.56
   495.6 2256.91     506 2255.47   510.7 2255.87   516.5 2258.39   537.4  2274.6
   559.8 2286.29   595.9 2297.37   618.6 2306.25   641.9 2312.02   656.9 2317.72
#Mann= 6 ,-1,0
       0      .1       0      10     .06       0   276.1     .07       0
   308.5    .045       0  326.84     .07       0  430.75      .1       0
#XS Ineff= 2 , 0
                          348.09         2270.26
Permanent Ineff=
       F       F
Bank Sta=308.5,326.84
XS Rating Curve= 0 ,0
Exp/Cntr(USF)=0,0
Exp/Cntr=0.3,0.1

Type RM Length L Ch R = 1 ,802     ,107.3,106,104.3
XS GIS Cut Line= 4
2195560.98758005 621927.728764062195776.56526715621730.216246275
2195978.89516341621523.0689715252196042.72542831621414.677955668
#Sta/Elev= 30
       0 2333.34      63 2306.84    69.2 2303.28    74.8 2298.47    80.3 2294.95
    96.5 2293.56   118.2 2284.35   139.9 2277.53   163.6 2272.31   204.5 2267.28
   259.3  2261.9   281.5 2260.95   287.2 2259.18   297.5 2253.44  306.352250.133
   318.3 2249.35  331.222250.133   338.1 2253.08   355.1 2255.02   388.9 2255.32
   394.9 2253.93   423.5 2253.41     456 2256.38   545.4 2255.12   575.7 2256.36
   584.3 2258.91     616 2271.65   660.2 2296.41   689.4  2308.6707.7314  2314.4
#Mann= 9 ,-1,0
       0      .1       0      80     .06       0     220      .1       0
     250     .06       0  306.35    .045       0  331.22     .06       0
  352.38      .1       0  382.38     .07       0  522.38      .1       0
Bank Sta=306.35,331.22
XS Rating Curve= 0 ,0
Exp/Cntr(USF)=0,0
Exp/Cntr=0.3,0.1

Type RM Length L Ch R = 1 ,696     ,56.1,57.4,59.2
XS GIS Cut Line= 3
2195618.79612184621975.9025488862195845.21291052621816.929058961
2196116.19045017 621436.35615884
#Sta/Elev= 30
       0 2322.98    11.5 2313.03    16.3 2310.77      31 2310.14    34.5 2309.18
    79.9 2290.28   102.2 2282.22     130 2274.51     163 2268.56   260.7 2258.53
   281.8 2251.48   288.7 2250.22   301.5 2249.71   307.82247.962   315.6 2246.57
  327.612247.963   353.2  2251.1   433.5 2251.38   453.1 2253.27   531.7 2253.47
   591.2 2255.14   599.8  2258.7   614.2 2267.62   634.8  2283.1   644.6 2286.84
   664.3 2291.74   688.7 2306.24   728.1 2321.61   734.6 2322.86743.8414 2326.28
#Mann= 10 ,-1,0
       0      .1       0      10     .06       0     130      .1       0
     250     .05       0   307.8    .045       0  327.61     .05       0
  346.65      .1       0  396.65     .06       0  466.65     .07       0
  566.65      .1       0
Bank Sta=307.8,327.61
XS Rating Curve= 0 ,0
Exp/Cntr(USF)=0,0
Exp/Cntr=0.3,0.1

Type RM Length L Ch R = 1 ,638     ,21.2,20.8,21
XS GIS Cut Line= 5
2195632.26929192622024.8309981092195741.74421794 621970.63549018
2195842.54786269621886.0904978112195978.03663251  621758.1890991
2196160.13353915621459.029895333
#Sta/Elev= 30
       0 2322.74    11.6 2320.57    26.5 2315.86   107.1 2282.95   130.5 2275.85
   187.4 2265.83   241.3 2262.02   266.7 2259.28   300.8 2251.98   340.4 2248.79
  347.12 2246.54   354.1 2245.19   360.2 2245.41     363 2246.58   368.7 2248.75
   374.4 2249.36   441.2 2250.36     460 2249.81   559.6 2251.56   591.1 2252.48
   614.1 2254.71   622.8 2254.69   642.6 2262.03   651.9 2266.82   670.7 2278.74
     681 2286.39   690.3 2291.59   731.6 2306.68     769 2322.94   790.3 2330.47
#Mann= 9 ,-1,0
       0     .06       0     100      .1       0  222.16     .06       0
  293.72     .05       0  347.12    .045       0     363     .05       0
  433.72     .06       0  510.04     .08       0  550.04      .1       0
#XS Ineff= 2 , 0
           335.6 2255.53  374.87         2254.05
Permanent Ineff=
       F       F
Bank Sta=347.12,363
XS Rating Curve= 0 ,0
Exp/Cntr(USF)=0,0
Exp/Cntr=0.3,0.1

Type RM Length L Ch R = 1 ,618     ,77.2,75.5,73.3
XS GIS Cut Line= 5
2195653.01587451622033.4008424122195762.49080053621979.205334483
2195863.29444529621894.6603421142195998.78321511621766.758943403
2196180.88012175621467.599739636
#Sta/Elev= 30
       0 2320.68    70.5 2291.27    92.8 2283.06     113 2277.83   160.9 2270.15
   178.7 2264.15   239.2 2260.78   263.9  2258.3   297.8 2250.97   309.9 2249.62
   337.5 2248.31   343.42246.018   348.8 2244.78   354.9 2244.92   358.4 2246.01
   365.7 2248.92   372.4 2249.31   450.9  2249.5   498.1 2250.83   529.5 2250.78
   587.1  2252.3     612 2254.21   619.8 2256.05   627.4 2259.92   638.6  2269.7
   648.9 2275.75   666.3 2287.79   727.4 2307.09   768.2 2324.76   790.3 2332.69
#Mann= 9 ,-1,0
       0     .06       0      80      .1       0  202.16     .06       0
  303.72     .05       0   343.4    .045       0   358.4     .05       0
  450.04     .06       0  470.04     .08       0  560.04      .1       0
#XS Ineff= 2 , 0
           323.5 2256.09  370.13         2255.04
Permanent Ineff=
       F       F
Bank Sta=343.4,358.4
XS Rating Curve= 0 ,0
Exp/Cntr(USF)=0,0
Exp/Cntr=0.3,0.1

Type RM Length L Ch R = 1 ,542     ,71.8,72.2,72.6
XS GIS Cut Line= 3
2195689.85245446622098.7457001912195930.72137859621967.472136541
2196235.42056761621509.821180699
#Sta/Elev= 30
       0 2314.12    16.3 2307.92    48.2 2298.09    70.1 2289.61   102.9 2279.84
   134.8 2273.26     165 2269.19   187.2  2264.5   244.1 2257.73   253.2 2254.77
   271.4 2246.71   366.4 2246.32  373.72 2244.37   382.8 2243.35  392.89 2244.38
     402 2247.11   464.5 2248.94     479  2248.1   493.3 2250.02   591.5 2250.95
   605.9 2253.62   613.5 2253.29   618.3 2255.15   630.6 2263.03   649.2 2270.56
   661.5 2276.99   673.9 2285.22   680.7 2287.88   752.8 2305.56824.1238 2327.57
#Mann= 8 ,-1,0
       0     .06       0      40      .1       0  284.32     .05       0
  373.72    .045       0  392.89     .05       0  424.32     .06       0
  524.32     .08       0  604.32      .1       0
Bank Sta=373.72,392.89
XS Rating Curve= 0 ,0
Exp/Cntr(USF)=0,0
Exp/Cntr=0.3,0.1
